--- BERGOOCK.prj (project) ---

Proj Title=BERGOOCK
Current Plan=p01
Default Exp/Contr=0,0
English Units
Geom File=g01
Flow File=f01
Plan File=p01
BEGIN DESCRIPTION:
----------MODEL BY WOOD PLC 2022----------
AFH study
Randolph County, WV
HEC-RAS Version: RAS 6.2
Vertical Datum: NAVD88
Projection: NAD 1983 StatePlane West Virginia S FIPS 4702 (US Feet)
Terrain: 1-meter LIDAR (FEMA Region III 3DEP collected 2016-2018)
Land Use: 2019 NLCD
Hydrologic Method:
WV SIR2010-5033 regression equations
Additional Model Notes:
Stream begins outside of county boundary;
END DESCRIPTION:
DSS Export Rating Curves= 0
DSS Export Rating Curve Sorted= 0
DSS Export Volume Flow Curves= 0
DXF OffsetX= 0
DXF OffsetY= 0
DXF ScaleX= 0
DXF ScaleY= 0

--- BERGOOCK.p01 (plan) ---

Plan Title=Floodplain
Program Version=6.20
Short Identifier=Floodplain
Geom File=g01
Flow File=f01
Subcritical Flow
K Sum by GR= 0
Std Step Tol= 0.01
Critical Tol= 0.01
Num of Std Step Trials= 20
Max Error Tol= 0.3
Flow Tol Ratio= 0.001
Split Flow NTrial= 30
Split Flow Tol= 0.02
Split Flow Ratio= 0.02
Log Output Level= 0
Friction Slope Method= 1
Unsteady Friction Slope Method= 2
Unsteady Bridges Friction Slope Method= 1
Parabolic Critical Depth
Global Vel Dist= 0 , 0 , 0
Global Log Level= 0
CheckData=True
Encroach Param=-1 ,0,0, 0
Mapping Interval=1HOUR
Computation Time Step Use Courant=        0
Computation Time Step Use Time Series=    0
Computation Time Step Count To Double=0
Computation Time Step Max Doubling=0
Computation Time Step Max Halving=0
Computation Time Step Residence Courant=0
Run HTab= 0
Run UNet= 0
Run Sediment= 0
Run PostProcess= 0
Run WQNet= 0
Run RASMapper=-1
UNET Theta= 0
UNET Theta Warmup= 0
UNET ZTol= 0
UNET ZSATol= 0
UNET MxIter= 0
UNET Max Iter WO Improvement= 0
UNET MaxInSteps= 0
UNET DtIC= 0
UNET DtMin= 0
UNET MaxCRTS= 0
UNET WFStab= 0
UNET SFStab= 0
UNET WFX= 1
UNET SFX= 1
UNET Gravity=32.174
UNET 1D Methodology=Finite Difference
UNET DSS MLevel= 1
UNET Pardiso=0
UNET DZMax Abort= 0
UNET Use Existing IB Tables= 0
UNET Froude Reduction=False
UNET Froude Limit= 0
UNET Froude Power= 0
UNET D1 Cores= 0
UNET WindReference=Eulerian
UNET WindDragFormulation=Hsu (1988)
UNET D2 Coriolis=0
UNET D2 Cores= 0
UNET D2 Theta= 1
UNET D2 Theta Warmup= 1
UNET D2 Z Tol= 0.01
UNET D2 Volume Tol= 0.01
UNET D2 Max Iterations= 20
UNET D2 Equation= 0
UNET D2 RampUpFraction=0.1
UNET D2 TimeSlices= 1
UNET D2 Turbulence Formulation=Non-Conservative (original)
UNET D2 Eddy Viscosity=0.3
UNET D2 Transverse Eddy Viscosity=0.1
UNET D2 Smagorinsky Mixing=0
UNET D2 BCVolumeCheck=0
UNET D2 Cores=0
UNET D2 SolverType=PARDISO (Direct)
UNET D2 Minimum Iterations= 2147483647
UNET D2 Maximum Iterations= 2147483647
UNET D2 Restart Number= 10
UNET D2 Relaxation Coeff=1.3
UNET D2 SOR Precondition Iterations= 10
UNET D2 ILUT Maximum Fill= 8
UNET D2 ILUT Tolerance=1E-08
UNET D1D2 MaxIter= 0
UNET D1D2 ZTol=0.01
UNET D1D2 QTol=0.1
UNET D1D2 MinQTol=1
Write IC File= 0
Write IC File at Fixed DateTime=0
Write IC File at Sim End=0
Echo Input=False
Echo Parameters=False
Echo Output=False
Write Detailed= 0
HDF Write Warmup=0
HDF Write Time Slices=0
HDF Flush=0
HDF Compression= 1
HDF Chunk Size= 1
HDF Spatial Parts= 1
HDF Use Max Rows=0
HDF Fixed Rows= 1
Calibration Method= 0
Calibration Iterations= 20
Calibration Max Change=0.05
Calibration Tolerance=0.2
Calibration Maximum=1.5
Calibration Minimum=0.5
Calibration Optimization Method= 1
WQ AD Non Conservative
WQ ULTIMATE=-1
WQ Max Comp Step=1HOUR
WQ Output Interval=15MIN
WQ Output Selected Increments= 0
WQ Output face flow=0
WQ Output face velocity=0
WQ Output face area=0
WQ Output face dispersion=0
WQ Output cell volume=0
WQ Output cell surface area=0
WQ Output cell continuity=0
WQ Output cumulative cell continuity=0
WQ Output face conc=0
WQ Output face dconc_dx=0
WQ Output face courant=0
WQ Output face peclet=0
WQ Output face adv mass=0
WQ Output face disp mass=0
WQ Output cell mass=0
WQ Output cell source sink temp=0
WQ Output nsm pathways=0
WQ Output nsm derived pathways=0
WQ Create Restart=0
WQ Fixed Restart=0
WQ System Summary=0
WQ Write To DSS=0
Sorting and Armoring Iterations= 10
XS Update Threshold= 0.02
Bed Roughness Predictor= 0
Hydraulics Update Threshold= 0.02
Energy Slope Method= 1
Volume Change Method= 1
Sediment Retention Method= 0
Sediment TS Multiplier= 1
Warm Up Method= 0
XS Weighting Method= 0
Number of US Weighted Cross Sections= 1
Number of DS Weighted Cross Sections= 1
Upstream XS Weight=0
Main XS Weight=1
Downstream XS Weight=0
Number of DS XS's Weighted with US Boundary= 1
Upstream Boundary Weight= 1
Weight of XSs Associated with US Boundary= 0
Number of US XS's Weighted with DS Boundary= 1
Downstream Boundary Weight= 0.5
Weight of XSs Associated with DS Boundary= 0.5
Percentile Method= 0
Sediment Output Level= 3
Mass or Volume Output= 0
Output Increment Type= 1
Profile and TS Output Increment= 1
Transport Output Increment 1
XS Output Flag= 0
XS Output Increment= 10
Read HDF5 Sediment Hotstart= 0
Sediment Hotstart Type= 0
Write Gradation File= 0
Read Gradation Hotstart= 0
Write HDF5 File= 1
Write Binary Output= 1
Write DSS Sediment File= 0
DSS Sediment Output Type= 1
SV Curve= 0
Specific Gage Flag= 0
Subcell Erosion Methods= 0
Subcell Deposition Methods= 0
Advection Scheme= 1
Matrix Solver= 0
Implicit Weighting Factor= 1
Maximum Outer Loop Convergence Iterations= 5
Convergence Maximum Absolute= 0.001
Convergence RMSE= 0.0001
Grain Fractions Max Abs Error= 0.001
Max Subgrid Regions= 1
Max Subgrid Length Scale= 3.402823E+38
Initial Layer Thickness= 3.402823E+38
Min Layer Thickness= 3.402823E+38
Max Layer Thickness= 3.402823E+38
Number of Layers= 5

--- BERGOOCK.f01 (steady flow) ---

Flow Title=Flow
Program Version=6.20
Number of Profiles= 1
Profile Names=P100yr
River Rch & RM=BERGOOCK,Main,11462
     392
River Rch & RM=BERGOOCK,Main,9065
     461
River Rch & RM=BERGOOCK,Main,7471
     636
River Rch & RM=BERGOOCK,Main,5994
     711
River Rch & RM=BERGOOCK,Main,3957
     858
River Rch & RM=BERGOOCK,Main,330
     980
Boundary for River Rch & Prof#=BERGOOCK,Main            , 1
Up Type= 0
Dn Type= 3
Dn Slope=0.0397
DSS Import GetInterval= 0
DSS Import GetPeak= 0
DSS Import FillOption= 0

--- BERGOOCK.g01 (geometry) ---

Geom Title=Geometry
Program Version=6.20

River Reach=BERGOOCK        ,Main
Reach XY= 30
     2204786.679      538041.977     2204736.158      538095.102
 2204548.0854808537976.794317192     2204195.012      537984.685
     2203826.783      538114.373     2203413.762       538012.29
     2203124.179      538323.227     2202690.159      538449.974
     2202784.075      538935.727     2202496.575      539036.768
     2202349.179      539301.8732202337.85821932539539.199872886
     2202196.575      539639.6332202133.08718281539852.641085936
     2201722.318      540054.728     2201044.972      540095.248
     2200837.554      540332.082     2200398.087      540423.736
     2200027.498      540358.632     2199976.508       540565.98
     2199509.298      540199.853  2199263.405156540315.439358007
2199039.82551401540315.498780007     2198624.265      540604.521
     2197890.535      540719.375     2197811.948      541112.011
     2197456.218      541646.526     2197241.728      541821.201
2197212.44745451542011.060014527     2196683.798      542571.984

Type RM Length L Ch R = 1 ,11462   ,266,266,266
XS GIS Cut Line= 4
2204687.46757767537381.2817660152204678.45285724537865.793817326
2204776.16271684538162.7573175532204800.79975794538297.082315146
#Sta/Elev= 30
       0 3372.84    91.9  3358.5   143.9 3354.83   167.8 3354.95   195.9 3350.31
   219.9 3348.57     344 3343.59     376 3338.39     400 3341.79   424.6 3341.33
     456  3343.7     484 3338.77   509.2 3336.72   534.5 3339.22   572.4 3337.38
   593.4 3333.18   610.3 3334.86   648.2 3333.69   686.1 3323.92   704.1  3322.6
   715.6 3317.68   723.1 3316.56   728.2 3317.65   803.7 3326.18   811.9 3329.83
   832.2 3345.32   856.6 3353.11   885.1 3366.49   909.5 3372.61   933.8 3376.41
#Mann= 3, -1 ,  0
       0     0.1       0   715.6   0.045       0   728.2     0.1       0
Bank Sta=715.6,728.2
XS Rating Curve= 0 ,0
Exp/Cntr=0.3,0.1

Type RM Length L Ch R = 1 ,11196   ,177.8,177.8,177.8
XS GIS Cut Line= 2
2204471.10386292537484.1721699032204555.12331988538280.606605704
#Sta/Elev= 30
       0 3362.11    21.1 3358.83    37.2 3354.36    45.3 3354.04    81.5 3344.78
   121.7 3341.39   157.9 3334.27     186 3331.99   307.5 3330.48   334.9 3326.32
     367 3329.94   399.2 3330.86   427.4 3328.26   451.5 3329.32   467.6 3320.81
   483.7 3305.87  486.57 3305.07   495.7 3304.38  502.72 3305.08   519.9  3308.4
     536 3307.95   588.3 3311.54   604.3 3310.63   616.4 3314.84   636.5 3316.73
   652.6 3324.72   671.3 3329.54   708.9 3335.41   722.3 3340.42   800.9 3360.01
#Mann= 3, -1 ,  0
       0     0.1       0  486.57   0.045       0  502.72     0.1       0
Bank Sta=486.57,502.72
XS Rating Curve= 0 ,0
Exp/Cntr(USF)=0,0
Exp/Cntr=0.3,0.1

Type RM Length L Ch R = 1 ,11018   ,195.9,195.9,195.9
XS GIS Cut Line= 2
2204266.75780878537576.1101338352204406.70283747538298.663302133
#Sta/Elev= 30
       0 3362.12    78.5 3347.54   135.5 3333.91     183 3317.09   196.6 3309.99
   204.8 3307.28   225.2 3305.54   274.1 3316.05   290.4 3314.33   298.5 3315.53
   310.7 3313.13   343.3 3317.12   392.2  3318.3   396.3 3317.13   415.1    3303
   424.8 3301.98   435.6 3296.99   441.1 3296.08  451.59 3296.99   461.5 3299.63
     490 3302.26   518.5 3301.49   526.7 3303.06   604.1 3298.94   620.4 3305.94
   665.2 3340.98   671.1 3344.48   681.7 3348.59   722.2 3355.82     736 3360.12
#Mann= 3, -1 ,  0
       0     0.1       0   435.6   0.045       0  451.59     0.1       0
#XS Ineff= 2 , 0
                          537.68         3304.18
Permanent Ineff=
       F       F
Bank Sta=435.6,451.59
XS Rating Curve= 0 ,0
Exp/Cntr=0.3,0.1

Type RM Length L Ch R = 1 ,10822   ,254.6,254.6,254.6
XS GIS Cut Line= 2
2204107.01954941537601.4493285822204217.29508667538331.368360953
#Sta/Elev= 30
       0 3357.27    48.3 3349.23    71.1 3342.54   112.7 3335.46   188.9 3315.66
   222.3 3309.75   274.8 3295.06     291 3293.72   303.1 3290.07   319.3 3296.92
   327.6 3303.83   339.5 3306.66   343.6 3306.09   363.8 3292.95   379.5 3286.38
   396.2  3285.5   398.6 3286.34   408.3 3290.23   433.1  3292.2   485.2 3289.99
   497.3    3292   525.6 3291.54   537.8 3293.98   570.1 3296.22   584.2  3302.1
   606.5 3318.84   626.3 3330.22   667.2 3341.57   723.9 3352.69   738.2 3357.82
#Mann= 3, -1 ,  0
       0     0.1       0   379.5   0.045       0   398.6     0.1       0
Bank Sta=379.5,398.6
XS Rating Curve= 0 ,0
Exp/Cntr(USF)=0,0
Exp/Cntr=0.3,0.1

Type RM Length L Ch R = 1 ,10568   ,259.2,259.2,259.2
XS GIS Cut Line= 4
2203858.48759465537593.9813785862203900.47171771537962.032831384
2203960.00802484 538176.497835552204030.17375717538350.402086073
#Sta/Elev= 30
       0 3355.63    35.4 3350.11    79.7 3346.48   180.4 3328.73   256.9 3303.37
   300.7 3278.31   311.6 3276.95   321.3 3278.54   341.4 3274.63   345.4 3276.08
   362.2 3288.97   373.7 3286.84   386.2 3276.59   406.9 3273.67   427.7 3276.96
   440.1 3282.85   470.2 3280.03   486.5 3274.99   503.9 3274.95   539.8 3277.83
     545 3280.22   560.5 3292.46   568.8 3295.81     611 3298.48   639.8 3302.95
   662.8 3310.15   671.4 3315.37     680 3317.24   731.8  3338.2   780.5 3350.24
#Mann= 3, -1 ,  0
       0     0.1       0   486.5   0.045       0   503.9     0.1       0
#XS Ineff= 2 , 0
          438.99 3294.91
Permanent Ineff=
       F       F
Bank Sta=486.5,503.9
XS Rating Curve= 0 ,0
Exp/Cntr=0.3,0.1

Type RM Length L Ch R = 1 ,10308   ,189.4,189.4,189.4
XS GIS Cut Line= 4
2203746.43604661537601.4493285822203737.68401984537923.523913609
2203683.42145389538098.5644489492203847.95955711538420.639033976
#Sta/Elev= 30
       0 3357.67   199.8 3327.25   235.7 3316.13   259.8 3306.63   332.3 3290.56
   340.7 3286.66   361.6 3270.65     370 3266.54   386.7 3266.56   411.9 3263.04
   432.8  3263.6  440.61 3261.56   445.4 3260.53   455.8 3261.52   466.3 3266.22
   478.9 3279.79   487.3 3283.04   522.8 3280.28   558.5  3282.7   589.2 3282.62
   602.7 3284.41   647.8 3285.13     683 3290.76     697 3296.54   718.1 3298.85
   753.3 3314.61   768.9 3317.45   781.5 3322.85   822.8 3335.38   867.1 3344.71
#Mann= 3, -1 ,  0
       0     0.1       0  440.61   0.045       0   455.8     0.1       0
Bank Sta=440.61,455.8
XS Rating Curve= 0 ,0
Exp/Cntr(USF)=0,0
Exp/Cntr=0.3,0.1

Type RM Length L Ch R = 1 ,10119   ,279.7,279.7,279.7
XS GIS Cut Line= 4
2203312.88281263 537643.559403432203504.51526767537896.560246675
2203534.63699885538156.3278256122203714.98118545538448.835921623
#Sta/Elev= 30
       0 3377.12    49.2 3361.57    74.9 3355.15     112 3352.75   137.5 3347.69
   202.7 3324.93     263 3306.52   283.7 3297.55   308.1 3293.29   317.4 3292.91
   339.3 3287.74   350.4 3287.26   362.3 3284.52   406.6 3257.42   425.9 3253.68
   434.8 3252.85     446 3253.75   475.1 3259.48   547.5 3261.67   589.4 3268.63
   631.6 3270.96   665.7  3271.1   731.8 3279.19     782 3293.57   795.7 3296.26
   847.7 3315.34   859.7 3316.44   868.4 3320.84     890 3327.87   922.5 3336.75
#Mann= 3, -1 ,  0
       0     0.1       0   425.9   0.045       0     446     0.1       0
Bank Sta=425.9,446
XS Rating Curve= 0 ,0
Exp/Cntr=0.3,0.1

Type RM Length L Ch R = 1 ,9839    ,255.8,255.8,255.8
XS GIS Cut Line= 4
2203104.03728191 537806.246754932203191.55754958538070.557963295
2203405.10700269 538191.335932682203573.14591662538523.912949828
#Sta/Elev= 30
       0 3361.28    53.7 3347.36    78.9 3344.66   129.5 3334.37   179.7 3318.79
   196.9 3316.78   208.2 3313.67   222.2 3306.29   264.3 3290.32   292.9 3284.22
   306.7 3276.84   325.1 3261.59   338.9 3253.15   384.8 3249.85     394    3245
   404.1 3244.12     417 3243.11  422.76  3244.1   430.8 3249.41   435.4 3250.26
   465.7 3247.21   485.9 3248.08   500.9 3256.02   511.3 3257.74   584.1 3258.26
   649.5 3263.79   735.8 3286.76   772.3  3293.3   839.5 3316.79   896.4 3332.66
#Mann= 3, -1 ,  0
       0     0.1       0   404.1   0.045       0  422.76     0.1       0
Bank Sta=404.1,422.76
XS Rating Curve= 0 ,0
Exp/Cntr(USF)=0,0
Exp/Cntr=0.3,0.1

Type RM Length L Ch R = 1 ,9584    ,229.7,229.7,229.7
XS GIS Cut Line= 4
2202977.28637474537862.6065698032203088.28363373538226.344039748
2203183.00653726 538412.563619492203415.84864626 538641.86694839
#Sta/Elev= 30
       0 3371.05    23.6 3363.84    61.2 3356.52    86.3 3349.68   103.1 3343.19
   111.4 3341.84   132.3 3332.85   157.4 3326.34   178.3 3317.38   186.7 3315.73
   215.5 3303.65   229.2 3301.81   279.9 3282.53   366.5 3253.43   401.4 3245.69
   428.4 3242.36   471.6 3233.58   482.2  3232.5   489.4 3233.59   504.6 3239.26
   549.5 3238.79   578.7 3234.79   601.5 3237.15   624.4 3250.26   638.6 3252.59
   695.1 3268.71   706.5 3270.18   723.4 3277.24   823.8  3307.7     916 3330.35
#Mann= 3, -1 ,  0
       0     0.1       0   471.6   0.045       0   489.4     0.1       0
#XS Ineff= 2 , 0
                          546.68         3244.36
Permanent Ineff=
       F       F
Bank Sta=471.6,489.4
XS Rating Curve= 0 ,0
Exp/Cntr=0.3,0.1

Type RM Length L Ch R = 1 ,9354    ,288.5,288.5,288.5
XS GIS Cut Line= 4
2202750.45540052537972.535263504 2202844.9772896538310.363496712
2203044.52349989538558.9210568962203275.57700654538770.720104658
#Sta/Elev= 30
       0 3354.83       9 3353.57    50.5 3338.09     171 3306.84   199.4 3298.19
   212.5 3291.56     225 3289.97   270.7 3269.11   303.9 3256.55   316.3 3249.58
   375.1 3231.58   423.4 3226.25   441.6 3227.08   452.4 3223.36   472.4 3222.52
   482.7 3221.55   490.8  3222.5   508.3 3225.07     523  3224.2   539.1 3228.01
   559.6    3226   625.4 3229.15   642.5 3236.21   679.4 3241.58   726.2 3253.74
   812.5 3281.45   826.4 3283.56   891.9 3303.81   962.1 3313.08     983 3317.29
#Mann= 3, -1 ,  0
       0     0.1       0   472.4   0.045       0   490.8     0.1       0
Bank Sta=472.4,490.8
XS Rating Curve= 0 ,0
Exp/Cntr(USF)=0,0
Exp/Cntr=0.3,0.1

Type RM Length L Ch R = 1 ,9065    ,256.5,256.5,256.5
XS GIS Cut Line= 4
2202306.11942099538370.0325677922202573.40650873 538483.24184296
2202738.42535151538490.5470409892203190.05474211538867.273073485
#Sta/Elev= 30
       0 3299.44    16.2  3296.9   123.9 3266.39   132.6 3262.44   149.9 3250.25
   167.3 3245.39   184.7 3244.08   210.7 3246.83   229.8 3246.08   249.8 3242.24
   271.6 3242.79   341.1 3229.65   357.1 3224.91  383.27 3213.06   389.1 3211.03
   397.1  3213.1   405.2 3212.81   421.2  3216.2   437.2 3223.31   475.6 3226.54
   594.9 3226.32   666.1 3229.25   684.4 3227.89   753.9 3235.33   817.1 3257.96
   830.6 3260.53   874.4 3275.78   884.9  3277.3   940.4 3297.69  1043.6  3320.8
#Mann= 3, -1 ,  0
       0     0.1       0  383.27   0.045       0   397.1     0.1       0
Bank Sta=383.27,397.1
XS Rating Curve= 0 ,0
Exp/Cntr=0.3,0.1

Type RM Length L Ch R = 1 ,8809    ,212.3,212.3,212.3
XS GIS Cut Line= 4
2202300.60122469538518.661733767 2202638.4294579538749.715240417
2202879.98539667538697.2030798152203125.04214615538902.000506164
#Sta/Elev= 30
       0 3286.84    44.7 3276.18    81.9 3270.21   153.3 3247.86   167.4 3245.37
   198.2 3233.78   251.5 3223.58   309.4 3220.46   394.2 3212.24   427.4 3211.11
   441.5 3207.88   472.5 3208.27   498.6 3206.29   541.6 3200.56   550.2 3199.62
  563.66 3200.64   582.7 3204.83   599.4 3216.82   611.6 3220.78   619.8 3221.64
   652.6 3219.53   662.3 3220.69   743.8 3247.52   792.3 3258.09   846.9 3279.37
   854.8 3281.11   872.4 3289.85   891.3 3296.87   924.7 3305.51   975.8 3314.57
#Mann= 3, -1 ,  0
       0     0.1       0   541.6   0.045       0  563.66     0.1       0
Bank Sta=541.6,563.66
XS Rating Curve= 0 ,0
Exp/Cntr(USF)=0,0
Exp/Cntr=0.3,0.1

Type RM Length L Ch R = 1 ,8597    ,374.1,374.1,374.1
XS GIS Cut Line= 3
2202321.42146855538748.4809617872202842.35423692538950.589231629
2202991.31273016539051.562079368
#Sta/Elev= 30
       0 3258.02    37.3 3247.89    52.7 3245.64   140.2 3220.22   183.2 3213.94
   200.3 3207.01   213.2 3207.19   234.6 3211.14     256 3209.18   293.2 3199.53
   307.6 3197.95   320.5 3200.64   333.7 3196.65   344.8 3195.45   401.4 3198.06
   423.4  3194.2   478.7 3196.19   491.1 3194.24   513.5 3193.31   518.9 3194.32
   543.6 3212.32   547.8 3217.43     561 3238.45   570.6 3249.02   596.5 3258.57
   614.1 3267.75   628.2 3270.88   643.1 3278.87   676.9 3292.28   738.7 3305.04
#Mann= 3, -1 ,  0
       0     0.1       0   491.1   0.045       0   518.9     0.1       0
#XS Ineff= 2 , 0
          480.27 3212.19
Permanent Ineff=
       F       F
Bank Sta=491.1,518.9
XS Rating Curve= 0 ,0
Exp/Cntr=0.3,0.1

Type RM Length L Ch R = 1 ,8222    ,203.8,203.8,203.8
XS GIS Cut Line= 3
2202249.39137688538947.0522860942202579.74537923539152.637394852
2202850.55059145 539229.20012501
#Sta/Elev= 30
       0 3256.16    67.5 3235.09     111 3219.55   155.4 3205.77   170.6 3204.77
   178.1 3200.37   192.3 3197.16     233 3184.27   243.6 3182.85   250.4  3180.6
   257.7 3180.15   276.5 3179.22   281.2 3180.21     286  3182.5   295.4  3181.3
   309.5 3183.61   333.1 3182.98   346.2 3184.55   360.8 3184.75   370.8 3186.55
     402 3199.29   422.8 3209.94   460.2 3223.32   468.5 3224.67   547.5 3260.45
     560 3263.14   576.6 3270.45   601.5 3277.97   634.8 3285.37   670.5 3290.14
#Mann= 3, -1 ,  0
       0     0.1       0   257.7   0.045       0   281.2     0.1       0
Bank Sta=257.7,281.2
XS Rating Curve= 0 ,0
Exp/Cntr(USF)=0,0
Exp/Cntr=0.3,0.1

Type RM Length L Ch R = 1 ,8019    ,254.6,254.6,254.6
XS GIS Cut Line= 3
2202163.81114697539109.1114385642202507.55520694539360.478670193
2202831.21348501539390.581441506
#Sta/Elev= 30
       0 3264.89      69 3245.56   117.7  3225.2   149.1 3213.72   162.8  3210.2
   174.9 3202.94   183.8 3194.79   196.6 3180.26   203.6 3176.02   233.4 3173.38
   244.1 3176.39  256.44 3174.27  273.94 3174.25   282.9 3176.62   292.3 3177.05
   303.7  3174.3   323.7 3174.58   335.2 3172.91   338.9 3173.62   349.5 3181.82
     366 3184.68   393.2 3187.22   421.7    3183   434.5 3183.28   530.9  3227.7
   575.1 3240.18   627.3 3262.34   647.4 3268.95   671.5 3275.29   750.9 3286.74
#Mann= 3, -1 ,  0
       0     0.1       0  256.44   0.045       0  273.94     0.1       0
#XS Ineff= 2 , 0
          244.66 3193.42
Permanent Ineff=
       F       F
Bank Sta=256.44,273.94
XS Rating Curve= 0 ,0
Exp/Cntr=0.3,0.1

Type RM Length L Ch R = 1 ,7764    ,292.8,292.8,292.8
XS GIS Cut Line= 4
2202106.19071491539318.5233101942202249.39137688539464.559628829
2202473.40825401539549.6293290042202817.94053972539514.183620598
#Sta/Elev= 30
       0 3248.39    99.5 3224.69   149.4 3207.24   162.8 3201.45   210.3 3167.01
   220.3 3162.25   233.2  3165.5   284.7 3167.39   288.8  3167.2  296.04 3162.72
   303.3 3161.98   311.7 3162.67   335.9  3166.5   348.7 3175.19   377.7 3172.74
   399.4 3179.46   442.9 3184.09   471.1 3190.02   491.2 3189.76   495.2 3191.27
   512.7 3203.48   531.4 3212.92   540.9 3215.38   559.5 3223.74   574.7 3227.24
   631.9 3247.86     644 3250.44   672.1 3260.42   716.4 3271.08   790.5  3280.7
#Mann= 3, -1 ,  0
       0     0.1       0  296.04   0.045       0   311.7     0.1       0
#XS Ineff= 2 , 0
           284.7    3170
Permanent Ineff=
       F       F
Bank Sta=296.04,311.7
XS Rating Curve= 0 ,0
Exp/Cntr(USF)=0,0
Exp/Cntr=0.3,0.1

Type RM Length L Ch R = 1 ,7471    ,261.3,261.3,261.3
XS GIS Cut Line= 4
 2201992.1234221539422.0208365672202099.10157323539665.891252577
2202293.70312522 539778.533751912202778.35502704539854.130269842
#Sta/Elev= 30
       0 3243.34    93.5 3215.59   112.6 3212.72   130.1 3206.49   186.9 3191.92
   248.1 3182.48   265.5 3178.56     290 3178.28   313.8 3160.54   335.6 3152.33
   345.6 3151.67  360.65 3152.32   378.5  3159.1   387.7 3156.62   407.1 3155.54
   447.8 3156.93   466.3 3159.56   480.3 3158.77   497.7 3166.85   513.9 3168.87
   558.4 3181.09   655.6 3200.33   708.2 3212.59   756.8 3226.19   796.8  3232.5
   841.8 3237.12   866.9 3242.19   886.3 3249.96   914.7 3258.87   981.7 3269.58
#Mann= 3, -1 ,  0
       0     0.1       0   335.6   0.045       0  360.65     0.1       0
Bank Sta=335.6,360.65
XS Rating Curve= 0 ,0
Exp/Cntr=0.3,0.1

Type RM Length L Ch R = 1 ,7210    ,184.9,184.9,184.9
XS GIS Cut Line= 3
2201897.76994948539463.1418004932202106.19071491540111.089350163
2202126.04031162540397.490674088
#Sta/Elev= 30
       0 3239.77    22.6 3233.69    38.5 3226.48    48.4 3224.96   149.2  3187.9
   191.2 3177.86     229 3182.18   300.5 3175.42   313.1 3172.28   325.7 3171.96
   346.9 3168.41   372.3 3167.79   384.5 3169.18   392.9 3166.24   413.6 3154.16
   430.7 3150.63  446.35 3143.83   464.3 3142.51  472.22 3143.83   486.8 3147.72
     498 3152.89   517.3 3155.93   548.4 3167.83   591.7  3181.4     603 3183.66
   611.4 3187.77   670.2 3207.22   840.2 3238.12   899.3 3250.73   967.7  3269.9
#Mann= 3, -1 ,  0
       0     0.1       0  446.35   0.045       0  472.22     0.1       0
Bank Sta=446.35,472.22
XS Rating Curve= 0 ,0
Exp/Cntr(USF)=0,0
Exp/Cntr=0.3,0.1

Type RM Length L Ch R = 1 ,7025    ,239.9,239.9,239.9
XS GIS Cut Line= 3
     2201674.912      539564.4022201947.39394125540140.863745225
2201972.09732981540410.335081716
#Sta/Elev= 30
       0 3231.22    77.8 3203.18   124.6 3191.24   178.8 3181.39   204.4 3175.05
   235.3 3171.22   255.7 3166.45   293.1 3166.66     341 3162.99   358.6 3164.98
   416.1 3159.65   421.2 3157.52   437.2 3143.33  441.61 3141.22   452.2  3140.5
   467.2 3141.18   479.2 3143.22   536.2 3146.01   567.2 3160.77   598.1 3188.18
   615.8 3201.52   629.1  3209.2   637.6 3211.16     658 3220.28   738.4 3238.05
   746.4 3241.42   786.6 3248.06   859.4 3268.66     883  3273.2   908.2 3281.35
#Mann= 3, -1 ,  0
       0     0.1       0  441.61   0.045       0   467.2     0.1       0
#XS Ineff= 2 , 0
                          482.97         3146.68
Permanent Ineff=
       F       F
Bank Sta=441.61,467.2
XS Rating Curve= 0 ,0
Exp/Cntr=0.3,0.1

Type RM Length L Ch R = 1 ,6785    ,258.9,258.9,258.9
XS GIS Cut Line= 3
2201568.39561743539564.2363573382201656.61604724540101.435760299
2201757.43939559540452.742114728
#Sta/Elev= 30
       0 3242.66   150.9 3207.78   199.6 3194.48   211.7 3192.54     228 3188.04
   240.1 3186.67   345.5 3166.01   398.2 3159.43   423.4 3150.79   446.8 3139.88
   483.3 3138.41   499.5 3134.55   503.6 3133.69   520.4 3134.56   527.9 3135.87
   536.8 3141.42   552.5 3154.83   569.1 3173.63   581.6 3183.91   586.3 3186.34
     603 3192.11   639.8 3198.95   718.9 3221.52   743.9 3231.58   752.2 3233.35
     798 3248.79   838.1 3265.79   868.7 3280.71     893 3290.58   909.9 3296.11
#Mann= 3, -1 ,  0
       0     0.1       0   499.5   0.045       0   520.4     0.1       0
Bank Sta=499.5,520.4
XS Rating Curve= 0 ,0
Exp/Cntr(USF)=0,0
Exp/Cntr=0.3,0.1

Type RM Length L Ch R = 1 ,6526    ,259.5,259.5,259.5
XS GIS Cut Line= 4
2201327.60167842539614.9785449742201388.76957677540007.587881616
 2201419.4661117540137.8421034682201555.94353674540483.287634921
#Sta/Elev= 30
       0 3238.47    54.9 3218.81      63 3217.27    99.4 3202.07   107.5 3200.25
   127.7 3192.68     167 3181.99   273.5 3161.58   370.6 3150.55   378.7 3147.87
     411  3130.6   427.7 3128.54   441.2 3124.51   452.4 3123.81  480.64 3124.54
   489.4 3129.66   505.8 3135.25   534.8 3140.98     552 3146.35   573.5 3156.19
   595.9 3169.62   625.1 3182.24   693.9 3200.91     724 3213.92   771.3 3228.62
   835.8 3254.07     853 3258.03   874.5 3267.06   883.1 3268.56   902.6 3276.31
#Mann= 3, -1 ,  0
       0     0.1       0   441.2   0.045       0  480.64     0.1       0
Bank Sta=441.2,480.64
XS Rating Curve= 0 ,0
Exp/Cntr=0.3,0.1

Type RM Length L Ch R = 1 ,6267    ,272.6,272.6,272.6
XS GIS Cut Line= 3
2201076.88179419539696.5670020562201180.85587218540210.135932745
2201377.77647444540559.866922356
#Sta/Elev= 30
       0 3244.22    29.2 3234.04    78.2 3221.98    98.6 3214.29   159.8  3183.2
   217.1 3158.99   253.7  3149.7   310.8 3141.51   327.1 3141.99   342.7 3139.67
   347.5 3137.22   363.8 3121.34     372 3115.44   385.8 3111.95   395.7 3111.01
   405.9 3111.99   416.9 3116.71   478.1 3118.46     523 3125.07     558 3138.92
   637.3 3174.12     656 3178.67   683.6  3182.2   715.7 3192.37   734.2 3202.11
   766.5 3215.48   793.7  3221.5   885.5 3256.96   908.5 3264.16   925.3 3271.61
#Mann= 3, -1 ,  0
       0     0.1       0   385.8   0.045       0   405.9     0.1       0
Bank Sta=385.8,405.9
XS Rating Curve= 0 ,0
Exp/Cntr(USF)=0,0
Exp/Cntr=0.3,0.1

Type RM Length L Ch R = 1 ,5994    ,228.1,228.1,228.1
XS GIS Cut Line= 3
2200839.42599706539798.2608365672200918.05056913540142.281573561
 2201185.3966649540626.410193415
#Sta/Elev= 30
       0 3236.62    15.3 3227.29    86.6 3193.78   175.3 3163.53   199.9 3156.96
   232.8 3151.32   294.3 3131.56   335.3 3125.64   360.8 3110.85     379 3109.69
   401.9 3112.19  436.83 3102.55   447.8 3101.29   456.6 3102.52   474.3 3103.25
   489.7  3109.9   509.7 3111.19   525.3 3118.77   539.3 3128.34   561.8 3139.18
   574.4 3141.71   589.6 3147.16   612.7 3158.06   657.8 3173.65   709.8  3188.2
   721.8 3189.13   753.7 3199.43   786.4  3207.5   849.7 3238.85   905.9 3256.01
#Mann= 3, -1 ,  0
       0     0.1       0  436.83   0.045       0   456.6     0.1       0
Bank Sta=436.83,456.6
XS Rating Curve= 0 ,0
Exp/Cntr=0.3,0.1

Type RM Length L Ch R = 1 ,5766    ,107.4,107.4,107.4
XS GIS Cut Line= 4
2200659.56765388 539862.610453882200755.66490779540199.738524946
2200787.17220415540413.9881402032200996.69572495540727.485738998
#Sta/Elev= 30
       0 3222.25     125 3167.99   181.5 3149.55   223.1 3139.53   235.6 3138.48
   277.2 3123.32   314.6 3116.16   339.6 3106.04   396.5 3099.66   408.6 3102.31
     445 3104.55   465.2 3101.49   477.3 3094.96   489.7 3093.57   497.6 3093.01
   514.4 3093.67   525.9 3096.55   549.7 3095.31   558.2 3096.74   570.9  3103.3
   593.2 3121.02   604.7 3127.33     672 3144.07   710.5 3157.98     749 3164.76
   806.7 3179.28   841.2 3192.86   867.2 3200.53   912.5 3224.12   944.2 3235.81
#Mann= 3, -1 ,  0
       0     0.1       0   489.7   0.045       0   514.4     0.1       0
#XS Ineff= 2 , 0
                          529.11         3103.52
Permanent Ineff=
       F       F
Bank Sta=489.7,514.4
XS Rating Curve= 0 ,0
Exp/Cntr(USF)=0,0
Exp/Cntr=0.3,0.1

Type RM Length L Ch R = 1 ,5659    ,101.9,101.9,101.9
XS GIS Cut Line= 4
2200631.88642765539871.4037638272200699.03268547 540201.72003215
 2200651.3805025540462.7240343342200866.89833003540752.969148795
#Sta/Elev= 30
       0 3218.99      48 3196.77    79.4 3184.39     112 3172.45   140.6 3164.24
   173.2 3151.36   206.8 3141.73   295.7 3121.42   324.3  3116.5   360.9 3098.22
   389.4  3099.5   409.7  3096.8     426 3097.99   442.2 3092.75   458.5 3094.18
   477.73092.854   495.1 3090.14   501.33090.834     548 3090.94   564.2 3095.28
   576.4 3096.36   592.7 3094.05   610.4 3095.84     644 3105.66   704.4 3140.65
     740 3155.31   771.5 3163.43     882 3182.59   936.4 3197.38   963.9 3208.73
#Mann= 3, -1 ,  0
       0     0.1       0   477.7   0.045       0   501.3     0.1       0
Bank Sta=477.7,501.3
XS Rating Curve= 0 ,0
Exp/Cntr(USF)=0,0
Exp/Cntr=0.3,0.1

Type RM Length L Ch R = 1 ,5557    ,212.5,212.5,212.5
XS GIS Cut Line= 4
2200506.50041681539903.1678583192200543.16031334540245.373703117
2200606.12833515540485.3960309362200816.82411699540774.734948266
#Sta/Elev= 30
       0 3216.82    26.2 3206.98    54.3  3193.6    86.5 3174.42   102.6 3169.71
     122 3156.28   142.8 3147.09     167 3143.37   187.1 3136.82   291.7 3115.21
   352.2 3093.44   372.9 3090.98   401.9 3092.72   411.2 3088.74   439.1 3084.64
   451.5 3083.43  461.77 3084.64   472.2 3088.46   488.7 3089.31   501.1  3092.7
   509.4 3097.26   534.2 3096.22   550.7 3091.17     584 3092.59   656.6 3121.57
   681.1 3136.23   719.6 3154.72   859.9 3179.08   908.7 3189.96   950.2 3202.55
#Mann= 3, -1 ,  0
       0     0.1       0   439.1   0.045       0  461.77     0.1       0
Bank Sta=439.1,461.77
XS Rating Curve= 0 ,0
Exp/Cntr=0.3,0.1

Type RM Length L Ch R = 1 ,5344    ,267.3,267.3,267.3
XS GIS Cut Line= 3
2200322.28204634539928.1456303122200383.72127424540481.098681453
2200547.55921532540816.651387701
#Sta/Elev= 30
       0 3202.19    45.3 3186.65   113.7 3153.43   145.9 3142.54     154 3141.43
   206.3 3125.34   274.7 3116.91   359.2 3097.21   371.3 3095.78   383.4 3098.39
   390.2 3098.03   399.5 3094.12   411.6 3086.03   419.6 3078.95   422.8 3078.38
   475.9 3078.04   492.5 3076.14   500.1 3075.75   508.1 3076.17   520.6 3076.83
   540.3 3088.68   552.4 3092.79   574.3 3095.77   592.1 3090.91   649.9 3097.28
   700.3 3112.56   761.2 3123.26   823.5 3132.11   876.9  3142.3   929.8 3149.63
#Mann= 3, -1 ,  0
       0     0.1       0   492.5   0.045       0   508.1     0.1       0
Bank Sta=492.5,508.1
XS Rating Curve= 0 ,0
Exp/Cntr(USF)=0,0
Exp/Cntr=0.3,0.1

Type RM Length L Ch R = 1 ,5077    ,346.2,346.2,346.2
XS GIS Cut Line= 4
2200224.69597531539945.3689100532200129.15999177540290.314724868
2200139.66281252540498.1564859622200349.01319342540849.997433275
#Sta/Elev= 30
       0 3177.58    12.3 3170.99    81.5 3158.05     179 3130.01   203.2 3128.84
   223.9 3130.82     253 3127.46   265.4 3122.11   276.5 3115.01   290.3 3110.09
   302.8 3103.39   311.1 3101.54   319.4 3097.43   340.2  3093.9   360.8 3086.91
   404.9 3067.18   412.6 3065.32   424.9  3064.4  434.79  3065.3   472.9    3073
     513 3069.57     521 3072.17     529 3072.28   565.1    3084   630.1 3087.22
   676.6 3093.12   793.9 3112.84   886.1 3122.79   904.7 3127.21   975.5 3137.91
#Mann= 3, -1 ,  0
       0     0.1       0   412.6   0.045       0  434.79     0.1       0
Bank Sta=412.6,434.79
XS Rating Curve= 0 ,0
Exp/Cntr=0.3,0.1

Type RM Length L Ch R = 1 ,4731    ,294.7,294.7,294.7
XS GIS Cut Line= 4
2200084.36750741539955.1282331752199887.28936867540360.627137345
2200016.31174727540618.6718945442200023.40088895540810.078719939
#Sta/Elev= 30
       0 3178.13      37 3167.77   131.3 3145.97   206.9 3122.21   246.9 3113.58
   282.5 3103.79   295.8 3096.54   326.9 3084.22   366.8 3069.81   375.6 3067.99
   393.9 3066.44   450.9 3065.92   500.7 3068.04   529.4 3070.96   545.4 3070.78
   571.2 3066.92   609.9 3064.46   636.8 3057.97   668.4  3053.6     684 3052.63
  693.82 3053.56   715.3 3075.31   732.2 3086.36   781.9 3102.46   801.9  3112.1
   809.9 3112.97   821.9 3119.19   841.9 3126.15     914 3146.78   930.9  3153.9
#Mann= 3, -1 ,  0
       0     0.1       0   668.4   0.045       0  693.82     0.1       0
Bank Sta=668.4,693.82
XS Rating Curve= 0 ,0
Exp/Cntr(USF)=0,0
Exp/Cntr=0.3,0.1

Type RM Length L Ch R = 1 ,4436    ,191.9,191.9,191.9
XS GIS Cut Line= 4
     2199930.901      539917.6092199874.87843801540241.643229107
2199705.60426083540476.8588500882199705.29811699540754.066433275
#Sta/Elev= 30
       0 3185.24    11.7  3179.8      28 3175.37    44.2 3168.01    52.3 3166.86
      97  3149.2   113.2 3145.48   157.9 3127.42   202.5 3111.53   275.6 3093.41
   316.2 3077.52   367.7 3064.34   442.2 3062.92   447.9  3059.9   466.3 3044.32
   473.7 3041.37     486 3040.34  495.23 3041.33   505.3 3044.76   525.2 3047.94
   559.5 3043.63   574.7  3048.7     627 3054.55     647 3061.28     707 3075.58
     751 3088.33     791 3104.12     831  3118.1   869.8  3135.5   895.8 3142.97
#Mann= 3, -1 ,  0
       0     0.1       0   473.7   0.045       0  495.23     0.1       0
#XS Ineff= 2 , 0
                           527.8         3070.77
Permanent Ineff=
       F       F
Bank Sta=473.7,495.23
XS Rating Curve= 0 ,0
Exp/Cntr=0.3,0.1

Type RM Length L Ch R = 1 ,4244    ,287.2,287.2,287.2
XS GIS Cut Line= 3
2199829.19285828539877.7339561342199540.90109658540416.508723912
2199583.43594666540767.815078341
#Sta/Elev= 30
       0 3185.25    40.2 3177.49   121.9 3149.04   171.7  3128.5   245.6 3102.67
   278.1 3083.89   307.4 3071.32   344.2 3063.33   366.8 3062.68   380.4 3060.03
   393.4 3050.31   412.2 3039.48   425.9 3036.91     443 3036.06  454.25 3036.84
   466.6 3043.34   502.9 3045.28   557.4 3041.72     571 3036.08   611.1 3039.87
   627.8 3049.88   656.1 3051.04   696.3 3063.19   736.8 3071.03     781 3082.77
     793 3087.62   857.5 3105.72     906 3127.84   934.1 3136.09   964.9 3140.81
#Mann= 3, -1 ,  0
       0     0.1       0   425.9   0.045       0  454.25     0.1       0
#XS Ineff= 2 , 0
                          501.08         3055.68
Permanent Ineff=
       F       F
Bank Sta=425.9,454.25
XS Rating Curve= 0 ,0
Exp/Cntr(USF)=0,0
Exp/Cntr=0.3,0.1

Type RM Length L Ch R = 1 ,3957    ,152.5,152.5,152.5
XS GIS Cut Line= 4
2199715.14297248539830.5707724872199363.19513161540026.404057602
2199400.69362777540476.3725869992199476.70840381540783.504214906
#Sta/Elev= 30
       0    3165   131.6 3135.49   186.4 3120.14   273.5 3085.76   296.4 3078.24
   346.7  3070.4   402.8 3071.01   441.7 3066.97   453.7 3063.65   513.9 3059.87
   521.9 3057.17   606.2 3051.89   610.3 3050.34   630.3 3033.65  644.84 3028.17
   662.4 3027.28     673 3028.13   682.5 3029.53   694.5 3036.32   702.5 3037.71
   718.6 3037.55   734.7 3031.84   742.7 3030.98   843.1 3029.36   850.9  3032.4
   879.8 3051.26   908.7 3064.92     987 3085.93  1032.3 3101.48  1170.7 3140.71
#Mann= 3, -1 ,  0
       0     0.1       0  644.84   0.045       0     673     0.1       0
#XS Ineff= 2 , 0
                          720.42          3041.5
Permanent Ineff=
       F       F
Bank Sta=644.84,673
XS Rating Curve= 0 ,0
Exp/Cntr=0.3,0.1

Type RM Length L Ch R = 1 ,3805    ,261.4,261.4,261.4
XS GIS Cut Line= 4
2199044.55819162539844.0775485052199211.72015246540012.515554853
2199250.68444569540493.9030009532199394.62000784540810.327559666
#Sta/Elev= 30
       0 3146.66    51.4 3130.49   148.1 3108.48   193.2 3091.13   209.6 3080.79
   235.3 3059.82   260.6 3051.45   275.5 3051.85   292.5 3056.64   338.6 3054.15
   366.4 3059.13   394.5 3054.84   458.7 3052.47   482.8 3049.05   522.9 3023.73
   535.4 3022.69     543 3022.16  559.23 3022.69   571.1 3030.09   623.2  3024.9
   671.4 3027.73   679.4 3031.15   691.5  3041.8   715.5  3041.4   737.1 3046.59
   776.6 3061.54   794.2 3064.46   820.5 3076.13   888.1 3087.45  1067.9  3132.2
#Mann= 3, -1 ,  0
       0     0.1       0   535.4   0.045       0  559.23     0.1       0
#XS Ineff= 2 , 0
                          586.77         3040.93
Permanent Ineff=
       F       F
Bank Sta=535.4,559.23
XS Rating Curve= 0 ,0
Exp/Cntr(USF)=0,0
Exp/Cntr=0.3,0.1

Type RM Length L Ch R = 1 ,3543    ,291.1,291.1,291.1
XS GIS Cut Line= 4
2198835.21159788539963.0239513242198957.12031746540302.330906879
 2199085.3916477540489.7565728382199138.97486138540856.627548147
#Sta/Elev= 30
       0 3173.73    36.3 3149.22    77.5 3138.41    87.3 3133.09   112.8 3123.84
   159.6 3099.85   189.3 3089.44   295.6 3058.42   350.8 3037.05   361.9 3030.79
   380.1 3017.34   412.5 3014.46     431 3014.02  435.38 3014.47   443.9 3015.98
     458 3024.69   491.4 3027.03   514.4 3023.71   543.2 3024.56     549 3025.75
   562.7 3034.46   596.7 3036.23   607.4 3039.85   627.5 3051.17   684.1 3058.64
     721 3067.46     866 3106.83   902.4 3119.63   926.6 3130.85   958.4 3139.04
#Mann= 3, -1 ,  0
       0     0.1       0   412.5   0.045       0  435.38     0.1       0
Bank Sta=412.5,435.38
XS Rating Curve= 0 ,0
Exp/Cntr=0.3,0.1

Type RM Length L Ch R = 1 ,3252    ,225.5,225.5,225.5
XS GIS Cut Line= 4
2198585.18181067540099.2866490322198694.92172389540428.506388711
2198819.97418315 540607.152759082198927.16200537 540922.33599823
#Sta/Elev= 30
       0 3145.17      61 3120.09    82.1 3113.92     124 3095.97   168.3 3090.98
   186.6 3081.46   200.2 3071.48   238.1 3054.49   313.8 3039.16   347.8 3036.79
   382.9 3037.69   394.4 3032.82   417.3 3016.04   437.4 3007.37   446.1 3006.01
   460.1 3004.98   469.9 3006.04   481.7 3010.38   503.5 3011.61   518.7    3016
   557.8 3018.68   579.5 3027.31   592.6 3035.78   622.2  3047.1   651.7 3063.09
     694 3065.99   736.2 3074.05   752.9 3080.39     797 3104.05     898 3140.09
#Mann= 3, -1 ,  0
       0     0.1       0   446.1   0.045       0   469.9     0.1       0
Bank Sta=446.1,469.9
XS Rating Curve= 0 ,0
Exp/Cntr(USF)=0,0
Exp/Cntr=0.3,0.1

Type RM Length L Ch R = 1 ,3027    ,248.1,248.1,248.1
XS GIS Cut Line= 3
     2198446.504      540165.017     2198560.084      540617.539
2198618.05549947540989.452315345
#Sta/Elev= 30
       0 3132.11    12.5 3124.23    66.2 3106.32    74.4  3101.9   105.4    3091
   169.3 3076.12   181.6 3068.89   214.6 3055.35   231.1 3046.64   272.4 3033.36
   313.6 3013.18   363.1 3005.76   420.8 3009.69     440 3005.02   449.9 2998.62
   466.2 2997.28   483.8 2998.52   493.1 3004.13   525.9  3029.1   539.1 3036.81
   571.4 3051.81   583.6 3054.19   595.7 3059.52   652.4 3074.31   700.9  3089.1
   713.1  3090.7   769.8 3106.28     782 3107.51   822.4 3116.43     843 3125.44
#Mann= 3, -1 ,  0
       0     0.1       0   449.9   0.045       0   483.8     0.1       0
Bank Sta=449.9,483.8
XS Rating Curve= 0 ,0
Exp/Cntr=0.3,0.1

Type RM Length L Ch R = 1 ,2779    ,250.4,250.4,250.4
XS GIS Cut Line= 3
2198229.99388464540210.7871233312198341.00984337540778.627372002
2198476.27066665541036.388563534
#Sta/Elev= 30
       0 3146.98    39.1  3120.8    79.9 3099.86    92.1 3095.77   115.6  3083.9
   149.2 3071.95   202.1 3056.91   235.7 3043.39   275.5 3032.01   316.3 3024.23
   324.4 3019.35   336.6 3008.83   352.9 3001.05   361.9 2999.37   397.8 2999.62
   406.2 2997.46  417.66  2991.1   436.9 2990.05   442.6 2991.05     463 2997.25
   479.3 3013.76   491.5 3022.94   503.8 3026.03   604.1  3033.8   665.8 3051.76
   676.3 3056.54   685.4 3057.15   714.5 3066.15   762.2 3084.95   869.7 3117.73
#Mann= 3, -1 ,  0
       0     0.1       0  417.66   0.045       0   442.6     0.1       0
Bank Sta=417.66,442.6
XS Rating Curve= 0 ,0
Exp/Cntr(USF)=0,0
Exp/Cntr=0.3,0.1

Type RM Length L Ch R = 1 ,2528    ,226.5,226.5,226.5
XS GIS Cut Line= 3
     2198004.293      540242.3662198082.71742955540787.481577593
     2198340.763      541103.127
#Sta/Elev= 30
       0 3131.44    63.5 3111.36    95.8 3098.65   144.3 3076.26   245.3 3042.88
   281.7 3032.65   342.3 3022.65   358.5 3017.09   395.2 2998.16   423.6 2991.52
   440.5 2983.43   459.5 2981.99   468.7  2983.4   479.7 2990.49   483.7 2991.08
   503.9 2993.31   540.3 2991.84     553 2993.29   567.2 2998.64   594.3 3017.43
   601.3 3020.23   614.9 3022.96   661.4 3026.03   718.3 3036.48   780.4 3053.29
   850.1 3075.14   878.4 3086.21   919.7 3094.97   950.7 3108.71   958.4 3109.94
#Mann= 3, -1 ,  0
       0     0.1       0   440.5   0.045       0   468.7     0.1       0
Bank Sta=440.5,468.7
XS Rating Curve= 0 ,0
Exp/Cntr=0.3,0.1

Type RM Length L Ch R = 1 ,2302    ,290.9,290.9,290.9
XS GIS Cut Line= 2
2197569.00231428 540491.517133912198301.45243279541144.852431258
#Sta/Elev= 30
       0 3157.86    32.5  3141.9    52.5 3135.03   122.7 3098.37   153.6 3089.05
   179.1 3076.62   186.5 3072.02   193.2  3065.1   224.8 3040.89   240.1 3026.02
   261.5 3001.63     283 2986.42   293.7 2983.69   369.1 2980.06   408.5 2978.83
   419.9 2980.02   438.4  2988.7   482.2 2991.21   496.4 2995.88   510.5 3004.52
   527.5 3011.76   545.6 3016.86   575.7 3020.85   645.5 3022.94   733.2 3038.05
   793.8 3054.06   867.8 3080.66   897.9  3087.3   935.5 3092.96   981.5 3109.58
#Mann= 3, -1 ,  0
       0     0.1       0   369.1   0.045       0   419.9     0.1       0
Bank Sta=369.1,419.9
XS Rating Curve= 0 ,0
Exp/Cntr(USF)=0,0
Exp/Cntr=0.3,0.1

Type RM Length L Ch R = 1 ,2011    ,282.1,282.1,282.1
XS GIS Cut Line= 4
2197356.96288685540858.634486076 2197667.9274024541027.907192181
2197909.82970123541014.3717741512198265.24159686   541175.903644
#Sta/Elev= 30
       0 3157.57    72.1 3116.13    81.1 3114.75   131.2 3091.57   172.3 3063.17
     204 3046.62   276.9 3025.33   299.7 3013.75   313.9 3004.25   349.8 2988.05
   386.3 2979.89   426.4 2978.29   458.5 2974.28   486.5  2974.5  515.24 2967.54
   526.6 2966.26  541.06 2967.51   550.4 2970.72   558.6 2977.41   578.6 2986.71
   612.1 2994.34   691.2 3021.35   713.1 3021.45   735.1 3027.34   752.7 3035.56
   796.5  3049.6   853.7 3073.55   890.2 3078.64   932.8 3088.38   986.7 3108.14
#Mann= 3, -1 ,  0
       0     0.1       0  515.24   0.045       0  541.06     0.1       0
Bank Sta=515.24,541.06
XS Rating Curve= 0 ,0
Exp/Cntr=0.3,0.1

Type RM Length L Ch R = 1 ,1729    ,202,202,202
XS GIS Cut Line= 2
2197276.78789418541008.3155624762198085.80074285541474.072170937
#Sta/Elev= 30
       0 3165.78    22.4 3154.82    97.9 3110.22   174.7 3074.14   197.8 3058.12
   220.8 3039.52   240.4 3031.44   257.8 3028.51   322.3 3010.36   386.6 3005.65
   398.6 2997.99   414.7 2981.49   431.1    2968   437.8 2964.76   456.2  2960.7
   465.5 2959.86  494.66 2960.69   539.3 2995.89     567  3007.7   603.9 3012.37
     627 3006.19   640.9 3005.01   719.3 3024.41   751.6 3039.64   779.3 3057.54
   793.2 3064.46   808.6 3076.24   857.8 3091.08   890.1 3114.28   933.5 3139.93
#Mann= 3, -1 ,  0
       0     0.1       0   456.2   0.045       0  494.66     0.1       0
Bank Sta=456.2,494.66
XS Rating Curve= 0 ,0
Exp/Cntr(USF)=0,0
Exp/Cntr=0.3,0.1

Type RM Length L Ch R = 1 ,1527    ,240.6,240.6,240.6
XS GIS Cut Line= 3
      2197145.92      541212.488     2197558.906      541399.609
     2197968.531      541617.552
#Sta/Elev= 30
       0 3164.47    81.5 3123.38   112.3 3110.87   134.2 3098.86   150.3 3094.19
   213.3 3058.84   222.8 3051.87   279.1 3023.72   327.4 3008.51     367  3004.1
     383 2997.02   424.1 2967.43  435.73 2956.58   459.4 2955.38     472 2956.57
   496.9 2959.51   536.4 2959.26   553.1 2964.69   603.4 2963.97   624.1 2965.06
   636.1 2967.75   671.4 2985.37   699.5 3005.51   735.8 3023.97   754.8 3040.95
   780.3 3058.09   814.4 3074.51   863.6 3104.67   875.5 3108.21   917.4 3127.08
#Mann= 3, -1 ,  0
       0     0.1       0  435.73   0.045       0     472     0.1       0
Bank Sta=435.73,472
XS Rating Curve= 0 ,0
Exp/Cntr=0.3,0.1

Type RM Length L Ch R = 1 ,1286    ,259.4,259.4,259.4
XS GIS Cut Line= 2
 2197037.4186679541332.7047332332197844.62814285541870.922322256
#Sta/Elev= 30
       0  3171.6    91.7 3123.91   114.8 3114.77   234.1 3056.43   260.4 3040.76
     285 3022.59   296.6 3016.05     334  2983.4   354.2 2970.45   368.6 2963.31
   394.6 2957.92     409 2952.25   433.5 2951.18   481.1 2954.51   505.6 2949.02
   522.5 2947.72  535.23 2948.95   548.8 2961.96   570.6 2979.44     585 2993.95
   596.5 2997.14   620.9 3008.88   639.8 3015.51   657.1 3025.03   666.8 3026.58
   691.7 3039.04   779.6 3058.73   849.5 3087.06   925.3 3122.27   970.2 3135.65
#Mann= 3, -1 ,  0
       0     0.1       0   505.6   0.045       0  535.23     0.1       0
Bank Sta=505.6,535.23
XS Rating Curve= 0 ,0
Exp/Cntr(USF)=0,0
Exp/Cntr=0.3,0.1

Type RM Length L Ch R = 1 ,1027    ,261.8,261.8,261.8
XS GIS Cut Line= 3
     2196922.936      541497.076     2197271.066      541781.151
     2197668.087      542063.466
#Sta/Elev= 30
       0 3165.86    86.2 3121.98   196.3 3072.69   218.4 3059.06   228.8 3056.81
   246.9 3045.79   259.6 3040.35     308 3003.84     332    2981   357.8 2968.01
   368.2 2960.19   373.4 2955.12   379.8 2945.75   418.9 2944.85   428.8  2942.7
   447.3 2941.34  457.79  2942.7     490  2948.1   544.8 2945.46   573.4  2956.9
   607.9 2960.32   622.5 2968.15   656.4 2990.62   670.3 2996.94   686.3 3007.21
     714  3020.1   746.2  3032.4   813.9 3068.93   882.6 3097.93   936.5 3115.32
#Mann= 3, -1 ,  0
       0     0.1       0   428.8   0.045       0  457.79     0.1       0
Bank Sta=428.8,457.79
XS Rating Curve= 0 ,0
Exp/Cntr=0.3,0.1

Type RM Length L Ch R = 1 ,765     ,186.1,186.1,186.1
XS GIS Cut Line= 2
2196753.88195107541748.8352502252197486.79779708542201.217979051
#Sta/Elev= 30
       0 3180.78    49.7 3152.96     139 3095.88   181.3 3072.75   204.8 3058.13
   243.2 3043.11   270.6 3028.35   341.1 2999.54   359.9 2989.89     389 2965.02
   425.7 2940.79   449.3  2935.9   468.1 2937.96   487.3 2935.84   518.5 2935.96
   533.7 2934.97   536.7 2936.01   543.3 2939.81   562.1 2938.57   585.6 2942.43
   613.8 2940.89   646.7 2942.62   670.2 2949.34   693.7 2959.93   717.2 2974.75
     736 2989.38   762.2 3014.09   787.7 3034.82   834.7 3058.63   861.3 3066.98
#Mann= 3, -1 ,  0
       0     0.1       0   518.5   0.045       0   536.7     0.1       0
Bank Sta=518.5,536.7
XS Rating Curve= 0 ,0
Exp/Cntr(USF)=0,0
Exp/Cntr=0.3,0.1

Type RM Length L Ch R = 1 ,579     ,248.8,248.8,248.8
XS GIS Cut Line= 2
 2196720.1972328542000.2976785532197372.11270183542281.925445711
#Sta/Elev= 30
       0 3126.36    26.1 3116.73    65.3 3092.74      74  3089.5   113.2 3066.98
   137.6 3057.53   161.2 3046.61   226.6 3008.33   286.7 2981.28   301.9 2977.81
   318.1 2970.65     366 2938.47   374.7 2930.15  376.51 2929.52   383.4 2928.19
  406.77 2929.52   418.3 2933.12   440.1 2931.72   470.6 2934.53   508.8 2932.87
     549 2935.11   575.1 2933.49   605.6 2936.65   614.4 2940.99   640.5 2961.59
     658 2970.69   666.6 2977.24   679.7 2989.96   697.1 3003.41   710.1 3009.79
#Mann= 3, -1 ,  0
       0     0.1       0  376.51   0.045       0  406.77     0.1       0
Bank Sta=376.51,406.77
XS Rating Curve= 0 ,0
Exp/Cntr(USF)=0,0
Exp/Cntr=0.3,0.1

Type RM Length L Ch R = 1 ,330     ,,,
XS GIS Cut Line= 4
2196740.39769688542104.7920651372196785.30872944542216.521951032
2197019.72241161542436.6955497082197063.53805314 542664.53688565
#Sta/Elev= 30
       0 3084.22    30.6 3068.72      78 3050.34    99.6 3045.14   140.8 3038.47
   157.3 3032.03   165.4 3026.79   179.2 3012.52   203.2 2999.76   214.9 2997.47
   227.6 2989.23   244.1 2982.42   261.5 2970.45   270.1 2958.62   284.2 2926.68
     289 2921.65   295.5 2919.66   305.4 2918.39  316.13 2919.64   326.7 2922.03
   349.3 2922.03     420 2928.54   439.9 2931.64   446.6 2934.78   480.4 2957.96
   487.4 2961.38   507.7 2965.66   564.7 2972.25   627.3 2989.97674.0339  3009.2
#Mann= 3, -1 ,  0
       0     0.1       0   295.5   0.045       0  316.13     0.1       0
Bank Sta=295.5,316.13
XS Rating Curve= 0 ,0
Exp/Cntr(USF)=0,0
Exp/Cntr=0.3,0.1
LCMann Table=0

Chan Stop Cuts=-1
Use User Specified Reach Order=0
Composite Channel Slope=5
